--- TAYLORRN.prj (project) ---

Proj Title=TAYLORRN
Current Plan=p01
Default Exp/Contr=0,0
English Units
Geom File=g01
Flow File=f01
Plan File=p01
BEGIN DESCRIPTION:
----------MODEL BY WOOD PLC 2022----------
AFH study
Randolph County, WV
HEC-RAS Version: RAS 6.2
Vertical Datum: NAVD88
Projection: NAD 1983 StatePlane West Virginia S FIPS 4702 (US Feet)
Terrain: 1-meter LIDAR (FEMA Region III 3DEP collected 2016-2018)
Land Use: 2019 NLCD
Hydrologic Method:
WV SIR2010-5033 regression equations
Additional Model Notes:
None
END DESCRIPTION:
DSS Export Rating Curves= 0
DSS Export Rating Curve Sorted= 0
DSS Export Volume Flow Curves= 0
DXF OffsetX= 0
DXF OffsetY= 0
DXF ScaleX= 0
DXF ScaleY= 0

--- TAYLORRN.p01 (plan) ---

Plan Title=Floodplain
Program Version=6.20
Short Identifier=Floodplain
Geom File=g01
Flow File=f01
Subcritical Flow
K Sum by GR= 0
Std Step Tol= 0.01
Critical Tol= 0.01
Num of Std Step Trials= 20
Max Error Tol= 0.3
Flow Tol Ratio= 0.001
Split Flow NTrial= 30
Split Flow Tol= 0.02
Split Flow Ratio= 0.02
Log Output Level= 0
Friction Slope Method= 1
Unsteady Friction Slope Method= 2
Unsteady Bridges Friction Slope Method= 1
Parabolic Critical Depth
Global Vel Dist= 0 , 0 , 0
Global Log Level= 0
CheckData=True
Encroach Param=-1 ,0,0, 0
Mapping Interval=1HOUR
Computation Time Step Use Courant=        0
Computation Time Step Use Time Series=    0
Computation Time Step Count To Double=0
Computation Time Step Max Doubling=0
Computation Time Step Max Halving=0
Computation Time Step Residence Courant=0
Run HTab= 0
Run UNet= 0
Run Sediment= 0
Run PostProcess= 0
Run WQNet= 0
Run RASMapper=-1
UNET Theta= 0
UNET Theta Warmup= 0
UNET ZTol= 0
UNET ZSATol= 0
UNET MxIter= 0
UNET Max Iter WO Improvement= 0
UNET MaxInSteps= 0
UNET DtIC= 0
UNET DtMin= 0
UNET MaxCRTS= 0
UNET WFStab= 0
UNET SFStab= 0
UNET WFX= 1
UNET SFX= 1
UNET Gravity=32.174
UNET 1D Methodology=Finite Difference
UNET DSS MLevel= 1
UNET Pardiso=0
UNET DZMax Abort= 0
UNET Use Existing IB Tables= 0
UNET Froude Reduction=False
UNET Froude Limit= 0
UNET Froude Power= 0
UNET D1 Cores= 0
UNET WindReference=Eulerian
UNET WindDragFormulation=Hsu (1988)
UNET D2 Coriolis=0
UNET D2 Cores= 0
UNET D2 Theta= 1
UNET D2 Theta Warmup= 1
UNET D2 Z Tol= 0.01
UNET D2 Volume Tol= 0.01
UNET D2 Max Iterations= 20
UNET D2 Equation= 0
UNET D2 RampUpFraction=0.1
UNET D2 TimeSlices= 1
UNET D2 Turbulence Formulation=Non-Conservative (original)
UNET D2 Eddy Viscosity=0.3
UNET D2 Transverse Eddy Viscosity=0.1
UNET D2 Smagorinsky Mixing=0
UNET D2 BCVolumeCheck=0
UNET D2 Cores=0
UNET D2 SolverType=PARDISO (Direct)
UNET D2 Minimum Iterations= 2147483647
UNET D2 Maximum Iterations= 2147483647
UNET D2 Restart Number= 10
UNET D2 Relaxation Coeff=1.3
UNET D2 SOR Precondition Iterations= 10
UNET D2 ILUT Maximum Fill= 8
UNET D2 ILUT Tolerance=1E-08
UNET D1D2 MaxIter= 0
UNET D1D2 ZTol=0.01
UNET D1D2 QTol=0.1
UNET D1D2 MinQTol=1
Write IC File= 0
Write IC File at Fixed DateTime=0
Write IC File at Sim End=0
Echo Input=False
Echo Parameters=False
Echo Output=False
Write Detailed= 0
HDF Write Warmup=0
HDF Write Time Slices=0
HDF Flush=0
HDF Compression= 1
HDF Chunk Size= 1
HDF Spatial Parts= 1
HDF Use Max Rows=0
HDF Fixed Rows= 1
Calibration Method= 0
Calibration Iterations= 20
Calibration Max Change=0.05
Calibration Tolerance=0.2
Calibration Maximum=1.5
Calibration Minimum=0.5
Calibration Optimization Method= 1
WQ AD Non Conservative
WQ ULTIMATE=-1
WQ Max Comp Step=1HOUR
WQ Output Interval=15MIN
WQ Output Selected Increments= 0
WQ Output face flow=0
WQ Output face velocity=0
WQ Output face area=0
WQ Output face dispersion=0
WQ Output cell volume=0
WQ Output cell surface area=0
WQ Output cell continuity=0
WQ Output cumulative cell continuity=0
WQ Output face conc=0
WQ Output face dconc_dx=0
WQ Output face courant=0
WQ Output face peclet=0
WQ Output face adv mass=0
WQ Output face disp mass=0
WQ Output cell mass=0
WQ Output cell source sink temp=0
WQ Output nsm pathways=0
WQ Output nsm derived pathways=0
WQ Create Restart=0
WQ Fixed Restart=0
WQ System Summary=0
WQ Write To DSS=0
Sorting and Armoring Iterations= 10
XS Update Threshold= 0.02
Bed Roughness Predictor= 0
Hydraulics Update Threshold= 0.02
Energy Slope Method= 1
Volume Change Method= 1
Sediment Retention Method= 0
Sediment TS Multiplier= 1
Warm Up Method= 0
XS Weighting Method= 0
Number of US Weighted Cross Sections= 1
Number of DS Weighted Cross Sections= 1
Upstream XS Weight=0
Main XS Weight=1
Downstream XS Weight=0
Number of DS XS's Weighted with US Boundary= 1
Upstream Boundary Weight= 1
Weight of XSs Associated with US Boundary= 0
Number of US XS's Weighted with DS Boundary= 1
Downstream Boundary Weight= 0.5
Weight of XSs Associated with DS Boundary= 0.5
Percentile Method= 0
Sediment Output Level= 3
Mass or Volume Output= 0
Output Increment Type= 1
Profile and TS Output Increment= 1
Transport Output Increment 1
XS Output Flag= 0
XS Output Increment= 10
Read HDF5 Sediment Hotstart= 0
Sediment Hotstart Type= 0
Write Gradation File= 0
Read Gradation Hotstart= 0
Write HDF5 File= 1
Write Binary Output= 1
Write DSS Sediment File= 0
DSS Sediment Output Type= 1
SV Curve= 0
Specific Gage Flag= 0
Subcell Erosion Methods= 0
Subcell Deposition Methods= 0
Advection Scheme= 1
Matrix Solver= 0
Implicit Weighting Factor= 1
Maximum Outer Loop Convergence Iterations= 5
Convergence Maximum Absolute= 0.001
Convergence RMSE= 0.0001
Grain Fractions Max Abs Error= 0.001
Max Subgrid Regions= 1
Max Subgrid Length Scale= 3.402823E+38
Initial Layer Thickness= 3.402823E+38
Min Layer Thickness= 3.402823E+38
Max Layer Thickness= 3.402823E+38
Number of Layers= 5

--- TAYLORRN.f01 (steady flow) ---

Flow Title=Flow
Program Version=6.20
Number of Profiles= 1
Profile Names=P100yr
River Rch & RM=TAYLORRN,Main,13307
     370
River Rch & RM=TAYLORRN,Main,10616
     417
River Rch & RM=TAYLORRN,Main,9017
     475
River Rch & RM=TAYLORRN,Main,6316
     670
River Rch & RM=TAYLORRN,Main,6104
     760
River Rch & RM=TAYLORRN,Main,2900
     893
Boundary for River Rch & Prof#=TAYLORRN,Main            , 1
Up Type= 0
Dn Type= 3
Dn Slope=0.0242
DSS Import GetInterval= 0
DSS Import GetPeak= 0
DSS Import FillOption= 0

--- TAYLORRN.g01 (geometry) ---

Geom Title=Geometry
Program Version=6.20

River Reach=TAYLORRN        ,Main
Reach XY= 30
2347499.92844284703861.5148524052347153.24200001703507.313999996
     2347154.978703290.734000012     2346780.412703117.557000011
2346716.61000003702844.9880000052346493.08500002702845.422000021
2346369.82099998702474.762000009     2346012.617702500.370000005
     2345856.367702334.1369999952345644.99500002702322.851999998
       2345564.7702169.2060000152345351.06402281702185.556908876
2345154.97800003 701947.505000012344930.49800001702091.254999995
2344303.45000003701931.1850000022343531.05400002701471.212000012
2343475.23800002701339.7880000032342741.07196668701247.713029992
 2342290.4446823700554.5227152852342130.84000002699951.441000015
2341731.79217969699675.465535775     2341698.904699300.787000015
2341414.27400003699182.439999998     2341023.809698787.904000014
2340929.95999999698324.4640000162340226.24300003698166.774000019
2339938.05800003 697617.990000012339589.78400002697636.917999998
2339307.34200001697290.929000005      2338548.83697036.441000015

Type RM Length L Ch R = 1 ,13307   ,131.2,126.4,122.5
XS GIS Cut Line= 2
 2347571.5824182703806.7978819242347428.55410769703886.396246033
#Sta/Elev= 30
       0 2842.95     3.9 2839.18     8.5 2834.38    10.1 2832.92    13.1 2830.91
    22.2 2829.73    26.8    2828    31.4 2825.37    35.9 2821.98    40.5 2817.99
    45.4 2814.25    49.7 2811.75    54.3 2809.63    60.1 2805.21    62.5 2803.88
    63.4 2803.55      66  2803.3    72.6 2803.41    80.7 2802.56    86.3 2802.32
    90.9 2802.56    95.5 2802.75     100 2803.28   113.8 2805.39   121.9 2810.09
   128.3  2814.3   133.7 2816.81   141.2 2821.38   145.8 2823.43   163.7 2828.24
#Mann= 3 ,-1,0
       0      .1       0    80.7    .045       0    90.9      .1       0
Bank Sta=80.7,90.9
XS Rating Curve= 0 ,0
Exp/Cntr(USF)=0,0
Exp/Cntr=0.3,0.1

Type RM Length L Ch R = 1 ,13181   ,64.8,66.2,66.8
XS GIS Cut Line= 3
 2347474.7861816 703710.042520772347415.10886426703748.657255514
2347393.34419559703874.330664952
#Sta/Elev= 30
       0 2828.53     3.1 2828.84     5.8 2828.01     7.9 2826.96    17.4 2820.84
    21.5 2818.87    31.7 2814.53    44.7 2810.41    50.8 2808.69    56.2 2806.42
      65  2802.1    71.1 2799.47    77.5 2797.52   87.032795.376    91.9 2794.93
      96 2795.06    98.3 2795.38   104.1  2796.3   112.1 2797.15   116.3 2796.99
   119.1 2797.25   124.4 2798.44   129.4 2800.88   140.6 2807.78   152.8 2814.66
     165 2821.83     169 2823.91   173.1 2825.07   176.1 2825.63   198.6 2828.82
#Mann= 3 ,-1,0
       0      .1       0   87.03    .045       0    98.3      .1       0
Bank Sta=87.03,98.3
XS Rating Curve= 0 ,0
Exp/Cntr(USF)=0,0
Exp/Cntr=0.3,0.1

Type RM Length L Ch R = 1 ,13114   ,52.9,56.9,59.3
XS GIS Cut Line= 3
2347435.46936077703664.4069251642347361.04823562703717.063381633
2347316.81681219703839.928446726
#Sta/Elev= 30
       0 2820.62     5.8 2818.15    11.5 2816.32      23 2813.26    28.7 2811.52
    37.4 2809.32      53 2804.49    62.8 2802.06      66 2801.42    72.6 2799.64
    95.5 2794.91    99.8  2794.6   108.3 2794.54   116.8 2793.64   125.3 2791.09
   129.5 2790.74   136.4 2791.06   142.3  2791.4   145.1 2792.18   151.3 2794.51
   155.1 2796.81   163.6 2803.48   172.1 2810.53   176.3 2813.79   180.6 2816.43
   188.8 2822.41   193.3 2824.79   197.6 2826.32   201.8 2827.17   221.8 2829.11
#Mann= 3 ,-1,0
       0      .1       0   125.3    .045       0   136.4      .1       0
Bank Sta=125.3,136.4
XS Rating Curve= 0 ,0
Exp/Cntr(USF)=0,0
Exp/Cntr=0.3,0.1

Type RM Length L Ch R = 1 ,13058   ,81.4,82.9,84.7
XS GIS Cut Line= 2
2347419.75327902703627.9649072652347230.89212182703778.913415808
#Sta/Elev= 30
       0 2821.95     4.6 2819.47     9.7 2815.79    14.8 2813.77    21.2  2811.8
    40.4 2807.69    57.5 2804.69    68.9 2803.24    91.6 2799.69     103  2798.4
   111.6 2796.32   125.8 2790.97   131.5 2790.19   136.5 2790.38  142.04 2788.77
   145.7 2788.48   154.2 2788.78   158.2 2789.35   165.6 2789.38   168.5 2789.66
   174.2 2791.59   182.7 2795.47   188.9  2799.4   194.1 2801.68   196.9 2803.53
   214.5  2813.4   224.8 2818.59   228.2 2819.24     235 2819.53   241.8 2821.45
#Mann= 3 ,0,0
       0      .1       0  142.04    .045       0   154.2      .1       0
Bank Sta=142.04,154.2
XS Rating Curve= 0 ,0
Exp/Cntr(USF)=0,0
Exp/Cntr=0.3,0.1

Type RM Length L Ch R = 1 ,12975   ,96.3,93.5,90.4
XS GIS Cut Line= 2
2347398.96088428703600.5170913162347174.99542277703681.256991234
#Sta/Elev= 30
       0  2815.4       3 2814.23    24.2 2808.63    32.7 2805.85    45.5 2802.28
    49.7 2801.34    58.2 2799.95    84.5 2793.28   100.8 2790.28     105 2788.27
   117.8 2780.68     122 2779.93   126.3 2780.05   134.8 2779.05     139  2778.9
  142.532778.344   147.5 2777.79   151.8 2778.33   155.8 2779.21   162.1 2781.99
   168.8 2784.02     173 2784.44   177.3 2785.27   185.8 2789.21   190.7 2791.71
   198.6 2796.19   211.3 2802.23   215.6 2803.24   224.6 2806.08   238.1 2809.74
#Mann= 3 ,-1,0
       0      .1       0  142.53    .045       0   151.8      .1       0
Bank Sta=142.53,151.8
XS Rating Curve= 0 ,0
Exp/Cntr(USF)=0,0
Exp/Cntr=0.3,0.1

Type RM Length L Ch R = 1 ,12881   ,50.3,52.8,55
XS GIS Cut Line= 3
2347371.57952692703540.137687899 2347229.7581375 703549.26480702
 2347147.6140654703655.279806043
#Sta/Elev= 30
       0 2814.05     3.4 2813.02    15.4 2807.85    23.5 2805.63    35.5 2801.49
    51.5 2796.98    75.6 2792.29    99.6 2785.45   117.2 2782.55   119.7 2781.95
   127.7 2778.94   131.1  2778.2   143.2  2776.5   151.7 2774.71   160.3 2773.91
   167.3 2772.21   172.4 2771.83  178.642772.195   187.5 2772.27   191.7  2773.9
   197.4 2778.16     210 2789.21   212.8 2791.12   225.9 2798.15   229.6 2799.46
   243.2 2803.04   253.3 2804.11   263.5 2806.91   271.5 2810.14   276.2 2811.04
#Mann= 3 ,-1,0
       0      .1       0   167.3    .045       0  178.64      .1       0
Bank Sta=167.3,178.64
XS Rating Curve= 0 ,0
Exp/Cntr(USF)=0,0
Exp/Cntr=0.3,0.1

Type RM Length L Ch R = 1 ,12828   ,67.8,71,74.2
XS GIS Cut Line= 2
2347330.85853391703440.4414636512347079.51171504 703594.19831654
#Sta/Elev= 30
       0 2812.58     7.8 2808.94    19.9 2805.94    39.7 2797.83    47.4 2796.03
    59.4  2791.5    68.8 2788.67    82.9 2785.72   108.7  2781.7   129.8 2775.59
     148 2774.38   157.9  2772.1   167.3  2771.1   177.7 2767.42   181.3 2766.83
  191.342767.402   195.4 2769.07   200.3 2769.96   203.2  2771.5     216 2779.55
   223.3 2783.61   238.1  2794.9   242.3 2797.77     247 2800.09   255.6 2803.43
   267.2 2807.12   270.4 2807.84   279.8 2808.08   287.6  2810.7   294.6 2812.22
#Mann= 3 ,-1,0
       0      .1       0   177.7    .045       0  191.34      .1       0
Bank Sta=177.7,191.34
XS Rating Curve= 0 ,0
Exp/Cntr(USF)=0,0
Exp/Cntr=0.3,0.1

Type RM Length L Ch R = 1 ,12757   ,72.8,72.9,74.1
XS GIS Cut Line= 3
2347329.45436174703432.7185167032347222.03519055 703470.63116536
 2347050.7261855703477.652026223
#Sta/Elev= 30
       0    2814     1.4 2813.47     9.8 2808.71    22.6 2806.02      48  2795.8
    70.3 2789.51    86.2 2786.03    98.6 2781.17   104.8 2778.42   111.6  2776.3
   119.8 2774.27   131.8 2773.14   139.8 2771.26   145.1 2770.86   151.8  2769.7
   159.8 2769.84   171.8 2766.95   183.8  2763.5  187.282763.106   191.8 2762.77
   199.8  2763.1   203.8 2764.05   207.9 2765.89   215.9 2770.93   225.8 2778.33
   231.9 2782.36   241.2 2786.88   247.9 2789.17   263.5 2791.22   285.4 2795.26
#Mann= 3 ,-1,0
       0      .1       0  187.28    .045       0   199.8      .1       0
Bank Sta=187.28,199.8
XS Rating Curve= 0 ,0
Exp/Cntr(USF)=0,0
Exp/Cntr=0.3,0.1

Type RM Length L Ch R = 1 ,12685   ,99.2,98.8,99.3
XS GIS Cut Line= 3
2347314.00846784703370.9349411132347216.41850186703404.635073253
 2347050.7261855 703397.61421239
#Sta/Elev= 30
       0 2817.45    10.4 2814.43    18.9 2811.17    31.6 2804.62    35.8 2803.48
    44.3 2802.21    52.7 2798.05    69.3  2791.5    73.9  2789.4    86.6 2782.14
   100.7 2773.52   111.5  2767.6   115.5 2766.43   123.5 2765.61   143.5 2766.25
   155.5 2764.32   167.5 2764.24   175.1 2760.77   179.6 2759.98   191.6 2759.25
  193.772759.827   203.6 2762.78   207.6 2765.62   211.6 2769.19   215.6  2771.9
   227.6 2778.45   231.6 2779.91   235.6    2781   251.6 2783.61   269.1 2784.61
#Mann= 3 ,-1,0
       0      .1       0   179.6    .045       0  193.77      .1       0
Bank Sta=179.6,193.77
XS Rating Curve= 0 ,0
Exp/Cntr(USF)=0,0
Exp/Cntr=0.3,0.1

Type RM Length L Ch R = 1 ,12586   ,109.3,103.6,96.1
XS GIS Cut Line= 4
2347262.68233449703274.9439111782347182.58618684703306.120260531
2347081.76991859703306.8496499652347039.24309084703387.271357535
#Sta/Elev= 30
       0 2818.15       7 2815.78    11.3 2813.93    28.4  2801.5    32.7 2798.67
    41.3 2795.81    45.6 2792.78    54.2 2785.35    68.5 2774.18    88.4 2760.21
    96.4 2755.32   100.4 2753.32   105.4 2752.79   112.4 2752.43   116.4 2752.77
   120.4 2753.79   128.4 2757.03   136.4 2759.16   140.4 2759.51   160.4 2757.24
   176.4 2758.14   180.4 2758.73   193.9  2762.3   207.5 2764.51   213.4 2766.49
   222.2 2770.13   241.5  2775.7   248.2 2777.99   270.9 2782.95   277.7 2783.76
#Mann= 3 ,-1,0
       0      .1       0   105.4    .045       0   116.4      .1       0
Bank Sta=105.4,116.4
XS Rating Curve= 0 ,0
Exp/Cntr(USF)=0,0
Exp/Cntr=0.3,0.1

Type RM Length L Ch R = 1 ,12482   ,111,110.7,110.4
XS GIS Cut Line= 2
 2347121.5865207703166.2442563092347008.03926478703386.404584589
#Sta/Elev= 30
       0 2797.17     3.3 2794.37     7.8 2791.98    15.1 2790.61    18.1 2789.29
    25.8 2783.26    46.7  2765.2    53.7 2760.56    66.3 2749.98    70.8 2747.36
   76.892746.145    79.8 2745.84    95.3 2746.13    97.8 2746.43   102.3 2747.78
   111.3 2752.08   115.8 2753.39   120.3  2754.2     125 2755.76   129.3 2757.75
   133.8 2758.37   147.3 2758.81   151.8 2759.97   157.6 2762.92   169.8 2768.03
   178.8 2771.02   190.3 2773.98   214.8 2779.31   223.8 2779.99   247.7 2782.89
#Mann= 3 ,0,0
       0      .1       0   76.89    .045       0    95.3      .1       0
Bank Sta=76.89,95.3
XS Rating Curve= 0 ,0
Exp/Cntr(USF)=0,0
Exp/Cntr=0.3,0.1

Type RM Length L Ch R = 1 ,12371   ,108.8,107.4,106.8
XS GIS Cut Line= 3
2347037.50954494703135.0404302542346994.17089764703168.844575147
2346918.76165134703341.332391398
#Sta/Elev= 30
       0 2787.27      11 2788.15    16.9 2786.36      22 2782.86    27.1 2778.51
    37.2 2767.74    42.5 2762.57    47.3 2759.51    59.7 2753.15    67.3 2747.76
    72.8 2742.74   76.812740.332      78    2740    87.1 2740.33      99 2740.53
   103.3 2741.33   129.5 2749.82   138.3 2751.58   151.4 2754.91   160.1 2756.13
   166.1 2758.27   173.2 2762.04   177.6  2763.6   186.3 2764.19   190.7  2765.1
   199.1 2768.74   203.8 2770.12   219.7 2771.94   225.6 2773.19   243.2 2779.06
#Mann= 3 ,-1,0
       0      .1       0   76.81    .045       0    87.1      .1       0
Bank Sta=76.81,87.1
XS Rating Curve= 0 ,0
Exp/Cntr(USF)=0,0
Exp/Cntr=0.3,0.1

Type RM Length L Ch R = 1 ,12264   ,119.7,128.3,131.1
XS GIS Cut Line= 4
2346990.70380586703095.1688747382346894.49200886703102.969831252
2346888.42459823 703131.573338472346844.21917799703307.528246504
#Sta/Elev= 30
       0 2778.18     2.5 2777.17    14.6 2773.85    22.6 2770.37    38.7 2767.73
    54.7 2763.07      71  2759.2    86.8  2753.9     107  2748.9   115.1 2745.76
   123.3 2744.75   127.3  2743.7   143.2 2736.13  145.482735.701     148 2735.49
  158.872735.707   168.7 2736.39   176.7 2736.25     181 2736.64   185.2 2737.55
   192.5 2739.95   203.1 2744.24   218.2  2747.2   230.5 2754.06   255.8 2764.76
   263.5 2767.69   271.8 2769.65   276.4 2771.19   296.5 2778.87   307.2 2781.89
#Mann= 3 ,-1,0
       0      .1       0  145.48    .045       0  158.87      .1       0
Bank Sta=145.48,158.87
XS Rating Curve= 0 ,0
Exp/Cntr(USF)=0,0
Exp/Cntr=0.3,0.1

Type RM Length L Ch R = 1 ,12136   ,105.7,111.3,112.3
XS GIS Cut Line= 3
2346982.90284935703042.2957250332346851.15336156703057.030865115
2346679.53231825703155.842980957
#Sta/Elev= 30
       0 2780.29     2.7 2779.84    10.8 2775.27    18.8 2771.62    26.9 2769.86
    34.9 2767.02      43 2765.44      51 2762.88   104.1  2753.7   115.4 2749.56
   127.5 2742.35   134.9 2739.34   149.5 2736.08   163.7 2736.44     170 2735.68
   172.9 2735.04   182.2 2730.56   187.6 2730.15   205.2  2730.8  215.582728.932
   223.7 2728.26  229.582728.976   237.6 2732.06   253.1 2733.02   263.7 2732.24
   269.9 2734.04   292.6 2747.92   313.5 2762.29   325.3 2767.34   330.6 2770.75
#Mann= 3 ,-1,0
       0      .1       0  215.58    .045       0  229.58      .1       0
#XS Ineff= 2 , 0
          201.77 2735.49
Permanent Ineff=
       F       F
Bank Sta=215.58,229.58
XS Rating Curve= 0 ,0
Exp/Cntr(USF)=0,0
Exp/Cntr=0.3,0.1

Type RM Length L Ch R = 1 ,12024   ,186.8,180,171.4
XS GIS Cut Line= 3
2346956.89966097702980.7548458682346717.67032788 702999.82385068
2346639.66076274703078.700188765
#Sta/Elev= 30
       0 2776.56     8.8 2771.26    19.6 2765.99    36.8  2759.9    60.5 2754.05
      77 2752.79      85 2750.05      97 2747.82   109.3 2739.49   113.1 2738.12
   121.1 2736.74   133.1 2730.24   141.2 2727.17   145.2 2726.37   165.2 2725.25
   169.3  2724.3   173.3 2722.32   179.5 2721.64   186.9  2722.3   193.3 2724.46
   201.4 2723.28   209.4 2723.36   221.4 2726.07   237.5 2727.62   247.8 2730.68
   264.9 2732.95   281.9 2736.58   316.1 2746.47   337.5 2751.36   350.9 2755.41
#Mann= 3 ,-1,0
       0      .1       0   173.3    .045       0   186.9      .1       0
Bank Sta=173.3,186.9
XS Rating Curve= 0 ,0
Exp/Cntr(USF)=0,0
Exp/Cntr=0.3,0.1

Type RM Length L Ch R = 1 ,11844   ,206.4,210.9,213.3
XS GIS Cut Line= 4
2346757.54188339702759.7277446432346708.13582547702807.400256672
2346673.46490763702958.2187492732346592.85502365703052.697000385
#Sta/Elev= 30
       0 2731.07     7.9 2728.42    21.8 2726.63    29.7  2726.4    35.3 2725.26
    42.4  2722.9    51.9 2718.24    73.4 2715.12    86.9 2712.01    96.8 2711.36
   108.4 2711.36   116.8 2712.36   136.2 2712.48   144.4 2712.25   152.6 2710.72
   156.7 2711.03   164.9 2712.96   173.1  2716.6   193.7 2718.63   210.3 2720.94
   214.1 2721.73   222.3 2724.84   226.4 2725.88   248.3 2727.58   257.6 2729.22
   274.6 2733.93   297.4 2739.09   317.8 2744.72   332.5 2749.81   347.6 2756.21
#Mann= 3 ,-1,0
       0      .1       0    96.8    .045       0   108.4      .1       0
Bank Sta=96.8,108.4
XS Rating Curve= 0 ,0
Exp/Cntr(USF)=0,0
Exp/Cntr=0.3,0.1

Type RM Length L Ch R = 1 ,11634   ,90.3,91.8,92.6
XS GIS Cut Line= 2
2346687.33327477702718.1226432352346437.70266632702945.217155083
#Sta/Elev= 30
       0 2730.06    18.6 2726.53    49.7 2717.46    58.3 2714.74    69.9 2710.08
    75.9 2708.75      95 2707.35   103.5 2706.18   112.4 2704.38   117.5 2704.69
   128.6 2707.17   135.3 2708.12   154.5 2708.03     165  2706.8   188.8    2707
   200.7  2703.1   206.6 2703.04   213.9 2701.92   219.6  2701.6     226  2701.2
   231.4 2701.62   236.4 2704.85   247.6 2714.11   258.4 2723.69   273.4  2731.3
   281.9 2734.28   296.3 2736.46   304.5 2739.52   313.6    2742   337.5 2749.75
#Mann= 3 ,-1,0
       0      .1       0   219.6    .045       0   231.4      .1       0
#XS Ineff= 2 , 0
          201.12 2708.65
Permanent Ineff=
       F       F
Bank Sta=219.6,231.4
XS Rating Curve= 0 ,0
Exp/Cntr(USF)=0,0
Exp/Cntr=0.3,0.1

Type RM Length L Ch R = 1 ,11542   ,97,102.9,106.1
XS GIS Cut Line= 3
2346656.21717916702683.557606974 2346592.0911071702727.756976844
2346379.56232481702849.602889296
#Sta/Elev= 30
       0 2725.27     9.8 2723.83    19.5 2720.29    43.8 2713.86    58.3  2712.5
    72.9 2709.35    96.2 2702.48   100.8 2702.14   111.1 2703.76     121 2703.34
   128.5 2702.17   146.9 2697.83     158 2697.07   160.8  2697.3   165.4 2699.24
   169.7 2699.12   179.2 2695.61   193.1 2696.51   201.4 2696.31  221.282696.323
   229.9 2698.98   245.9  2698.8   248.4 2699.01   251.8  2700.4   260.6 2706.64
   278.1 2721.59   281.1 2723.54   285.3 2725.15   304.5 2727.92   322.9 2729.42
#Mann= 3 ,0,0
       0      .1       0   201.4    .045       0  221.28      .1       0
#XS Ineff= 2 , 0
          167.51 2701.41
Permanent Ineff=
       F       F
Bank Sta=201.4,221.28
XS Rating Curve= 0 ,0
Exp/Cntr(USF)=0,0
Exp/Cntr=0.3,0.1

Type RM Length L Ch R = 1 ,11439   ,94.2,91.4,89.6
XS GIS Cut Line= 3
2346624.08305122702634.9003396692346531.32927043  702693.7894718
2346363.20859597702716.310442457
#Sta/Elev= 30
       0 2725.31     9.4 2724.23    28.3 2720.83    42.5 2715.88    47.3 2714.56
    56.7 2713.01    68.2 2708.57    80.4 2705.07    93.8  2699.9   100.1 2698.17
   121.1 2694.38   129.2 2693.99   133.2 2694.62   137.3  2694.6  155.982689.476
   161.5  2688.9171.07382689.446   173.6 2689.59   181.7 2691.76   185.7 2691.87
   193.8 2690.68   205.9 2692.18     218 2692.78     222 2693.87   225.8 2695.89
   246.2 2708.86   254.3 2712.59   262.4 2714.06   274.5 2713.18   279.5 2713.46
#Mann= 3 ,-1,0
       0      .1       0  155.98    .045       0171.0738      .1       0
#XS Ineff= 2 , 0
                          183.68         2694.93
Permanent Ineff=
       F       F
Bank Sta=155.98,171.0738
XS Rating Curve= 0 ,0
Exp/Cntr(USF)=0,0
Exp/Cntr=0.3,0.1

Type RM Length L Ch R = 1 ,11347   ,92.4,92.5,92.5
XS GIS Cut Line= 2
2346598.89520758702517.7982615112346358.79910154702679.018029464
#Sta/Elev= 30
       0 2733.34    13.2 2728.97    24.6 2726.56    44.8 2721.27    51.5 2720.33
    61.1 2718.19    79.3 2712.56    93.8 2710.01    99.6 2709.68   104.5  2708.3
   113.7 2702.36   120.9 2696.29   125.5 2693.92   135.2 2692.27   165.8 2685.18
   171.1 2684.88  175.162685.187   181.5 2685.94     186 2687.07   191.2 2690.12
   194.6 2691.24   200.8 2691.68   209.1 2693.61   220.6 2694.63   224.9 2696.42
     235 2699.45   253.8 2706.64   263.5 2708.18   282.7 2707.63   289.2 2707.91
#Mann= 3 ,-1,0
       0      .1       0   165.8    .045       0  175.16      .1       0
Bank Sta=165.8,175.16
XS Rating Curve= 0 ,0
Exp/Cntr(USF)=0,0
Exp/Cntr=0.3,0.1

Type RM Length L Ch R = 1 ,11255   ,148.8,140.1,133.7
XS GIS Cut Line= 3
2346537.20762825702449.2955544362346391.11695807702546.333882806
2346358.05994511702640.173145405
#Sta/Elev= 30
       0 2730.18     3.5 2728.82       6 2727.09    23.7 2719.84    28.7  2717.2
    38.2 2714.48    41.1 2712.84    50.4  2706.1    73.3  2696.3    92.5 2688.94
    98.8 2684.77   102.1 2683.41   106.9 2682.32   111.7 2681.91   116.5 2682.18
   127.6 2683.68   140.5 2684.08   145.3 2683.75   153.6 2680.57   156.5 2680.12
   165.1 2680.64   169.3 2682.91   174.1 2687.46   179.9 2689.13   195.4 2690.84
   216.6 2691.89   230.1 2693.99   250.5 2695.39   267.7 2700.06   274.9 2701.65
#Mann= 3 ,-1,0
       0      .1       0   153.6    .045       0   165.1      .1       0
Bank Sta=153.6,165.1
XS Rating Curve= 0 ,0
Exp/Cntr(USF)=0,0
Exp/Cntr=0.3,0.1

Type RM Length L Ch R = 1 ,11115   ,99.9,99.9,105.1
XS GIS Cut Line= 4
2346307.32492699702371.2110081322346302.52057953702454.757680663
2346317.03889091702532.6246095992346344.62149139702648.313199233
#Sta/Elev= 30
       0 2728.06       6 2726.84      18 2723.58      26 2720.07      30 2716.73
      34 2712.28      38 2708.42      42 2705.32    50.3 2699.68    66.1 2689.95
    74.1 2686.03    78.1 2683.56    86.1 2676.22    89.6 2674.99    98.4 2674.68
  103.36 2674.99   110.6 2675.92   126.8 2675.81   147.2 2676.64   151.3 2677.89
   158.2 2681.15   167.6 2687.99   171.7 2689.91   175.8  2690.9   192.2 2691.53
   204.6 2693.11   208.7 2693.35   249.8 2695.04   266.3 2698.08   281.8 2703.41
#Mann= 3 ,-1,0
       0      .1       0    89.6    .045       0  103.36      .1       0
Bank Sta=89.6,103.36
XS Rating Curve= 0 ,0
Exp/Cntr(USF)=0,0
Exp/Cntr=0.3,0.1

Type RM Length L Ch R = 1 ,11015   ,151.7,152.3,153.4
XS GIS Cut Line= 2
2346221.00942983702367.0796001122346223.60974866702634.045667475
#Sta/Elev= 30
       0 2718.79     6.1 2718.39    10.1 2717.47    26.1 2711.93    34.1 2710.11
    38.1 2708.55    54.1  2700.4    70.1 2688.91    78.1 2684.24    82.1 2682.69
    98.1 2677.85   118.1 2674.14   134.1 2672.37   142.1 2669.69  145.322669.187
   150.1 2668.58   158.1 2668.53   163.7 2669.18   170.1 2671.49   178.1 2672.19
   180.7 2673.18   186.1 2676.39   190.1 2679.56   194.1 2682.14   206.1  2683.5
   218.1 2686.68   234.1 2688.61   249.4 2689.37   258.1 2690.52     267 2692.53
#Mann= 3 ,-1,0
       0      .1       0  145.32    .045       0   163.7      .1       0
Bank Sta=145.32,163.7
XS Rating Curve= 0 ,0
Exp/Cntr(USF)=0,0
Exp/Cntr=0.3,0.1

Type RM Length L Ch R = 1 ,10863   ,129.2,133.3,141.3
XS GIS Cut Line= 2
2346084.05930436702374.8805566262346058.92288893702642.713396935
#Sta/Elev= 30
       0 2701.59    26.4 2698.63    42.5 2695.02    46.5 2693.25    54.5 2688.73
    62.6 2684.85    70.6 2679.37    75.5 2677.39    82.5    2674    86.5 2672.63
    94.7 2670.24   114.8  2668.3   118.8 2667.24   122.8 2665.65   130.9  2664.4
   137.9 2662.85   146.9 2662.27   153.4 2662.79     159 2663.81     163 2665.13
   175.1  2670.8   179.1 2672.11   187.1 2676.06   195.2 2676.31   199.2 2677.08
   203.2 2678.58   211.2 2680.95   239.3 2687.71   251.4  2691.6     269 2694.95
#Mann= 3 ,-1,0
       0      .1       0   137.9    .045       0   153.4      .1       0
Bank Sta=137.9,153.4
XS Rating Curve= 0 ,0
Exp/Cntr(USF)=0,0
Exp/Cntr=0.3,0.1

Type RM Length L Ch R = 1 ,10729   ,112.9,113.5,114.2
XS GIS Cut Line= 2
2346071.05771017 702369.679918952345820.56032878702561.236740012
#Sta/Elev= 30
       0 2701.12     5.8 2699.98    13.7 2696.98    18.8 2694.11    28.8 2686.98
      54 2674.88      65 2670.15    78.2    2666    84.4  2663.4    90.2 2663.15
    99.3 2664.62   114.4 2664.03   127.3 2661.93   141.5 2657.02   149.7 2656.43
   155.8 2656.92   161.5 2658.12   175.8 2657.86     195 2659.33   204.3 2662.71
   215.1 2667.94   220.2  2669.5   229.6 2670.61   235.3 2672.31   249.4 2672.54
   260.4 2674.31   270.5 2675.13   284.2 2677.36   295.7 2680.03   315.3  2683.1
#Mann= 3 ,-1,0
       0      .1       0   141.5    .045       0   155.8      .1       0
Bank Sta=141.5,155.8
XS Rating Curve= 0 ,0
Exp/Cntr(USF)=0,0
Exp/Cntr=0.3,0.1

Type RM Length L Ch R = 1 ,10616   ,113.7,107.6,99.4
XS GIS Cut Line= 3
2345982.64686968702306.4054938932345776.35490854702439.021754628
2345778.95522738 702555.16932939
#Sta/Elev= 30
       0 2692.27    18.3 2688.93    26.7 2686.43    38.5 2683.75    44.3 2681.93
    69.5 2670.03    84.8  2660.8      98 2655.28   105.1 2651.81     108  2650.8
   113.8  2649.9   119.6 2650.04   124.62650.809   131.3 2652.62     134 2652.93
   145.6 2652.53   159.9 2652.64   180.4 2654.31   197.5 2653.72   226.4 2653.82
   241.8 2655.48   245.2 2655.97   255.4 2659.57   263.4 2661.68   271.4 2665.14
   279.4 2665.22   287.4 2667.38   305.9 2670.56   347.4 2679.85   361.4 2683.48
#Mann= 3 ,-1,0
       0      .1       0     108    .045       0   124.6      .1       0
#XS Ineff= 2 , 0
                          136.66          2655.4
Permanent Ineff=
       F       F
Bank Sta=108,124.6
XS Rating Curve= 0 ,0
Exp/Cntr(USF)=0,0
Exp/Cntr=0.3,0.1

Type RM Length L Ch R = 1 ,10508   ,158.9,160,164.2
XS GIS Cut Line= 4
2345865.44918501702198.9352341612345802.15520198702285.564322439
2345787.60366039702376.5016050422345712.47751746702534.828662992
#Sta/Elev= 30
       0 2692.65      34 2684.46    47.4 2683.04      54 2681.27    71.2 2678.55
    79.8 2676.41    90.3 2670.91    99.8 2666.83   123.1 2650.63   127.2 2648.61
  136.292645.489   147.1 2644.84   154.1 2645.49   163.6 2646.47   179.8 2646.22
   183.9 2646.66   187.9 2647.71     196 2651.41   207.4 2652.61   222.3 2651.55
     240 2651.44   248.8 2651.53   257.7 2652.46   266.5 2655.75   275.4 2658.07
   288.7 2663.06   297.5 2662.95   313.6 2665.04   349.6 2671.63   374.6 2678.08
#Mann= 3 ,0,0
       0      .1       0  136.29    .045       0   154.1      .1       0
Bank Sta=136.29,154.1
XS Rating Curve= 0 ,0
Exp/Cntr(USF)=0,0
Exp/Cntr=0.3,0.1

Type RM Length L Ch R = 1 ,10348   ,165.8,163.2,163.7
XS GIS Cut Line= 2
2345742.33882762 702181.367084262345565.56752659702422.473518657
#Sta/Elev= 30
       0 2679.93    14.6 2676.46    38.6 2672.52    71.3 2666.13    74.2 2664.99
    78.7 2662.56    84.1 2658.82    90.1 2653.65    98.4 2648.69   105.1 2643.33
   108.9 2641.28   111.9 2640.48   124.5 2639.05   135.9 2640.06   143.6 2639.49
   161.7 2639.24   167.4  2638.2   173.1 2637.57   178.3 2637.59  180.692638.215
   187.4 2640.73   190.3 2641.21   213.2 2642.16   218.9    2643     223 2644.48
   233.2 2649.34   252.7 2652.97   260.7 2656.57   292.4 2665.57     299 2668.22
#Mann= 3 ,-1,0
       0      .1       0   167.4    .045       0  180.69      .1       0
Bank Sta=167.4,180.69
XS Rating Curve= 0 ,0
Exp/Cntr(USF)=0,0
Exp/Cntr=0.3,0.1

Type RM Length L Ch R = 1 ,10185   ,104.2,101.3,97
XS GIS Cut Line= 3
2345646.73802196702117.6332138212345591.42183252702144.088782682
2345484.99829415702391.207846366
#Sta/Elev= 30
       0 2674.29     8.2 2667.33    22.6 2658.29    29.4  2653.2    37.6 2648.09
    51.6 2637.19    58.6 2633.17    60.5 2632.34    71.2 2630.08    89.8  2629.9
    97.3 2629.34  101.962629.879   113.3 2632.95   119.1 2633.51   136.5 2633.16
   149.6 2632.16   152.9 2631.02   155.9 2630.59   162.7 2630.67   171.2 2632.02
   180.8 2634.47   213.8 2635.06   231.3 2634.55   250.3  2637.2   261.7 2641.02
   275.9 2647.56     299 2659.95   308.2 2663.78   320.3  2670.6   330.4 2675.24
#Mann= 3 ,-1,0
       0      .1       0    89.8    .045       0  101.96      .1       0
#XS Ineff= 2 , 0
                          132.17            2641
Permanent Ineff=
       F       F
Bank Sta=89.8,101.96
XS Rating Curve= 0 ,0
Exp/Cntr(USF)=0,0
Exp/Cntr=0.3,0.1

Type RM Length L Ch R = 1 ,10084   ,114.4,115.3,118.3
XS GIS Cut Line= 4
2345533.09932844702052.0955545952345475.37808729702115.829425034
2345488.60587172702261.9363167022345447.11872964702379.783850721
#Sta/Elev= 30
       0 2657.78      23 2651.74    43.1 2645.53    69.4 2636.78    82.4 2633.75
    95.4 2627.83    99.4 2626.91   103.4 2626.66   115.5 2626.74   119.5 2625.88
   126.3 2622.68   127.5 2622.25   135.2 2621.91   139.6 2621.94  145.18 2622.75
   155.6 2625.45   159.6 2626.02   195.8 2626.61   203.8 2628.16   219.9 2629.65
   231.6 2632.36   240.4 2635.03   248.9 2635.91   265.8 2639.36   285.8 2644.24
     304 2651.38   316.7 2655.69   325.2 2657.45   332.8 2660.31   357.6 2668.33
#Mann= 3 ,-1,0
       0      .1       0   126.3    .045       0  145.18      .1       0
Bank Sta=126.3,145.18
XS Rating Curve= 0 ,0
Exp/Cntr(USF)=0,0
Exp/Cntr=0.3,0.1

Type RM Length L Ch R = 1 ,9969    ,83.8,87.3,94.9
XS GIS Cut Line= 4
2345515.66270351702034.6589296642345418.85937199702102.000377675
2345386.99243678702125.4496318932345343.70150591 702308.23356221
#Sta/Elev= 30
       0 2659.06      14 2655.68    43.2 2645.37    47.4 2644.38    62.7 2639.23
    76.2 2635.98    96.8 2629.57   131.2 2626.96     145 2627.29   156.4 2626.69
   161.3 2625.85   173.7 2622.27   194.2 2620.29   198.3 2619.24   202.4 2617.48
   206.5 2616.52   223.4 2616.81   231.2 2616.31   239.1 2616.83   247.6 2617.77
   251.8 2619.39     260 2626.29   264.1  2628.3   268.2 2630.85   284.6 2645.05
   292.9 2650.06   305.2 2653.11   309.2 2653.63   321.6 2653.75   345.3 2656.11
#Mann= 3 ,-1,0
       0      .1       0   223.4    .045       0   239.1      .1       0
#XS Ineff= 2 , 0
                          245.76         2620.81
Permanent Ineff=
       F       F
Bank Sta=223.4,239.1
XS Rating Curve= 0 ,0
Exp/Cntr(USF)=0,0
Exp/Cntr=0.3,0.1

Type RM Length L Ch R = 1 ,9881    ,99.7,99.6,99.1
XS GIS Cut Line= 3
2345493.35000922702015.6150996242345244.58617372702179.435186415
2345217.36499793702252.556008571
#Sta/Elev= 30
       0 2655.37    54.7 2637.78    68.5 2633.78    87.6 2629.46    97.3 2628.21
   111.7 2625.23   143.5  2623.5     169 2619.41   183.9 2619.74     193  2619.1
   197.8 2617.91   204.1  2613.1     207 2611.52   221.7 2610.88   227.2 2610.47
  234.992610.885   250.3 2613.15   255.2 2613.29     260 2612.39   264.8 2612.75
   274.4 2615.36   287.9 2614.29   297.9 2616.27   308.3 2619.53   310.5 2620.85
   329.6 2636.32   338.1 2640.68   346.7 2642.49   359.5 2643.08   375.9 2644.95
#Mann= 3 ,-1,0
       0      .1       0   221.7    .045       0  234.99      .1       0
#XS Ineff= 2 , 0
                          255.44          2615.3
Permanent Ineff=
       F       F
Bank Sta=221.7,234.99
XS Rating Curve= 0 ,0
Exp/Cntr(USF)=0,0
Exp/Cntr=0.3,0.1

Type RM Length L Ch R = 1 ,9782    ,182.5,171.4,166.5
XS GIS Cut Line= 3
 2345394.9748123701927.6257164982345368.10485098701970.964363797
2345140.14356618 702136.51799648
#Sta/Elev= 30
       0 2650.21    15.9 2644.48    29.3 2639.09    48.9 2632.51    60.8 2628.02
    70.7 2627.71    80.6 2625.34    88.8 2624.64   125.1 2619.19   135.6 2617.19
   143.3 2614.41   158.5 2610.44   169.6 2609.41   175.7 2608.12   192.9 2606.67
   198.52605.558   209.1 2605.02     214 2605.46     219 2608.09   223.9 2608.93
   248.6  2610.3   258.5  2611.4   284.5 2611.21   288.2 2612.35   298.8 2618.04
   304.5 2622.25   311.5 2628.14   318.9 2633.04   322.8 2634.11   332.7 2634.02
#Mann= 3 ,-1,0
       0      .1       0   198.5    .045       0     214      .1       0
Bank Sta=198.5,214
XS Rating Curve= 0 ,0
Exp/Cntr(USF)=0,0
Exp/Cntr=0.3,0.1

Type RM Length L Ch R = 1 ,9610    ,158.2,151.3,148.5
XS GIS Cut Line= 2
2345128.00874494701869.5519291172345130.60906378702143.452180048
#Sta/Elev= 30
       0 2640.15     7.6 2638.24    11.6 2636.68    19.6 2632.16    31.6 2627.01
    43.9 2620.28    47.6 2617.69      52 2612.66    59.6 2600.87   62.292598.277
    63.6    2597    67.6 2596.84    72.1 2597.07    79.6  2598.3    83.6 2599.22
    91.6 2599.16   103.6 2599.91   115.6 2605.53   123.6 2607.91   135.6  2608.5
   147.6 2607.71   163.6 2608.08   167.6 2608.85   175.6 2614.14   203.6  2625.1
   207.6 2626.42   227.6 2630.27   247.6  2632.7   255.6  2633.2   273.9 2632.38
#Mann= 3 ,-1,0
       0      .1       0   62.29    .045       0    79.6      .1       0
Bank Sta=62.29,79.6
XS Rating Curve= 0 ,0
Exp/Cntr(USF)=0,0
Exp/Cntr=0.3,0.1

Type RM Length L Ch R = 1 ,9459    ,89.6,93.1,95.4
XS GIS Cut Line= 3
2345023.12921848701906.8231657942344989.32507358701999.567871014
2345102.00555656702157.320547184
#Sta/Elev= 30
       0 2625.52     6.8  2622.7      11 2620.31    19.5 2618.03    32.3 2613.95
    57.9 2608.16    63.4 2606.38    66.4 2605.81    70.6 2606.42    74.9 2605.93
    83.4 2603.42   104.8 2599.56   117.4 2592.75   130.2 2588.34   135.1    2588
   150.7 2588.36   154.8 2589.71   169.5  2596.9   184.3 2597.67   194.1 2598.85
     200 2600.13   206.8 2603.44   218.7 2608.02   233.8 2618.14   241.3 2621.22
   248.1 2622.56   261.9 2623.72   267.8 2624.62   287.5 2629.38   292.6  2629.9
#Mann= 3 ,-1,0
       0      .1       0   130.2    .045       0   150.7      .1       0
Bank Sta=130.2,150.7
XS Rating Curve= 0 ,0
Exp/Cntr(USF)=0,0
Exp/Cntr=0.3,0.1

Type RM Length L Ch R = 1 ,9366    ,107.5,111.7,115.6
XS GIS Cut Line= 3
2344958.98802047701895.5551174962344925.18387558701965.763726121
2344955.52092869702183.323735563
#Sta/Elev= 30
       0 2618.09     6.5 2617.28    21.3  2613.6    41.8 2610.21    55.1 2606.37
      64 2605.16      71 2602.62    77.9 2598.18    81.4 2596.65    89.4 2596.23
   105.6 2596.98   126.1 2594.93   136.8 2594.85   154.1 2591.78   162.1 2589.73
   170.2 2589.35   182.8 2585.82     197 2584.32   204.1 2583.98   210.6 2584.24
   218.7 2588.03   226.8 2594.39   234.8 2599.35     251 2611.99     255 2614.55
   263.1 2617.28   271.2 2624.12   275.2 2626.83   283.3 2629.78   297.6 2633.42
#Mann= 3 ,-1,0
       0      .1       0     197    .045       0   210.6      .1       0
Bank Sta=197,210.6
XS Rating Curve= 0 ,0
Exp/Cntr(USF)=0,0
Exp/Cntr=0.3,0.1

Type RM Length L Ch R = 1 ,9254    ,118.4,118.3,117.6
XS GIS Cut Line= 2
2344925.18387558701875.6193397392344787.36697717702159.920866021
#Sta/Elev= 30
       0 2615.13     6.2 2613.04    19.5 2607.27    28.4 2604.38    48.2 2599.95
    55.1    2599      64 2596.97    73.8 2595.85    99.5 2591.42   126.2 2588.78
   139.5 2588.03     149 2586.45   166.6 2585.14   175.6 2583.39   187.5 2579.63
   197.3 2578.92   201.8 2579.05   204.42579.634   210.7  2581.1   219.5 2581.49
     224 2582.24   229.5 2584.18   232.9 2586.09   246.2 2595.55   277.3  2619.4
   290.7 2625.22   299.6 2626.54     304 2628.25   308.5 2630.99   315.9  2632.2
#Mann= 3 ,-1,0
       0      .1       0   187.5    .045       0   204.4      .1       0
Bank Sta=187.5,204.4
XS Rating Curve= 0 ,0
Exp/Cntr(USF)=0,0
Exp/Cntr=0.3,0.1

Type RM Length L Ch R = 1 ,9136    ,121,119.3,117.4
XS GIS Cut Line= 2
2344805.56920904701835.7477842232344681.62067776702120.916083452
#Sta/Elev= 30
       0 2613.15    11.3 2608.99    32.5 2596.66    40.8 2593.57    49.5 2590.96
      67 2587.98    80.1  2585.2    88.8 2582.25   110.6 2581.27   119.3 2581.63
   129.8 2580.88   145.5 2580.84   154.2 2579.43   180.4 2576.85   184.6 2575.56
   189.1 2575.22   199.8 2575.59   210.9 2577.72     215 2579.94   224.3 2586.32
   228.4 2589.56   241.4 2601.75   245.8 2605.46   251.4 2608.58   263.6 2612.47
     272 2614.31   284.9 2616.02   293.8 2615.91   302.5  2618.4   310.9 2619.66
#Mann= 3 ,-1,0
       0      .1       0   184.6    .045       0   199.8      .1       0
Bank Sta=184.6,199.8
XS Rating Curve= 0 ,0
Exp/Cntr(USF)=0,0
Exp/Cntr=0.3,0.1

Type RM Length L Ch R = 1 ,9017    ,107.7,103.3,98
XS GIS Cut Line= 2
2344664.28521884701799.3433204922344585.40888076702109.648035154
#Sta/Elev= 30
       0 2599.88    18.4 2595.01    26.7 2594.16    43.2 2590.89    55.5 2589.61
    76.2 2584.62    88.6  2582.3    96.8 2579.93     134 2576.44   146.3 2574.54
  153.462570.307   154.6 2569.58   158.7 2569.14     167 2569.08   171.1 2569.23
   172.7 2570.28   179.4 2573.84   183.5 2573.99   208.3 2572.31   216.5 2572.76
   228.9 2577.08   245.1 2585.64   253.7 2589.56   278.4  2603.4   282.5 2604.11
   286.7 2604.19   290.8 2605.34   294.9 2607.74   311.4 2615.01   320.2 2615.25
#Mann= 3 ,-1,0
       0      .1       0  153.46    .045       0   172.7      .1       0
Bank Sta=153.46,172.7
XS Rating Curve= 0 ,0
Exp/Cntr(USF)=0,0
Exp/Cntr=0.3,0.1

Type RM Length L Ch R = 1 ,8913    ,110.8,113.7,117
XS GIS Cut Line= 3
 2344522.1344557701795.8762287082344511.73318035701926.758943552
2344569.80696773702113.981899884
#Sta/Elev= 30
       0 2598.38    25.4 2592.94    33.4 2592.48    45.4  2588.1    61.5 2583.77
    75.2 2581.38    81.6 2579.63    97.6 2579.69     122 2576.61   142.2 2575.28
   146.4 2574.13   149.6 2572.59     159 2566.48   163.1 2565.07   167.3  2564.5
   178.3 2565.03   192.5  2565.9   230.2 2563.49   234.3 2563.91   238.5 2565.59
   255.3 2575.84     271 2591.32   280.4 2599.22   284.6 2600.69   288.8 2601.17
     293 2602.84   301.3 2610.36   313.9 2616.21   318.1 2617.82   327.3 2618.25
#Mann= 3 ,-1,0
       0      .1       0   163.1    .045       0   178.3      .1       0
#XS Ineff= 2 , 0
                          192.56         2570.86
Permanent Ineff=
       F       F
Bank Sta=163.1,178.3
XS Rating Curve= 0 ,0
Exp/Cntr(USF)=0,0
Exp/Cntr=0.3,0.1

Type RM Length L Ch R = 1 ,8800    ,119.6,122.5,123.9
XS GIS Cut Line= 2
2344438.92425288701781.141088626 2344392.1185138702103.580624532
#Sta/Elev= 30
       0 2594.14    20.2 2593.37    32.4 2592.08    44.5 2588.06    56.6 2585.13
    84.9 2574.59   101.1 2571.08   109.2  2570.2   129.4 2570.75   137.5 2569.66
   141.5 2567.63   153.6 2557.55   155.62556.704   157.7 2555.85   164.8 2555.73
   177.9 2556.75   194.1 2555.62   202.1 2557.94   210.2 2558.42   226.4  2562.6
   238.5 2563.79   242.6 2564.87     246 2566.75   254.7 2573.42   266.8 2585.04
   278.9 2591.95     287  2595.2   288.4 2596.33   299.1 2607.33   325.8 2631.44
#Mann= 3 ,-1,0
       0      .1       0   155.6    .045       0   177.9      .1       0
Bank Sta=155.6,177.9
XS Rating Curve= 0 ,0
Exp/Cntr(USF)=0,0
Exp/Cntr=0.3,0.1

Type RM Length L Ch R = 1 ,8677    ,166.1,168.6,167.3
XS GIS Cut Line= 3
2344429.38975048701785.4749533562344331.44440758701820.145871196
2344254.30161539702048.107155989
#Sta/Elev= 30
       0 2593.12    26.7 2591.99      48 2589.38    60.3 2589.11      83 2585.03
   103.9 2580.34   113.4 2573.95   117.7 2571.89   126.1 2569.39   132.5  2565.4
   138.8 2562.46   151.5 2559.59   173.6 2559.06   201.5 2547.67   210.6 2546.87
     219 2546.87  224.792547.726   231.7 2549.68   244.3 2550.26   248.6 2551.29
   252.8 2554.24   265.1 2565.09   274.5 2574.84   278.1 2576.68   286.6 2578.53
   299.2 2588.97   309.2  2592.8   326.2 2604.21   338.7 2611.14   344.6 2613.36
#Mann= 3 ,-1,0
       0      .1       0   201.5    .045       0  224.79      .1       0
Bank Sta=201.5,224.79
XS Rating Curve= 0 ,0
Exp/Cntr(USF)=0,0
Exp/Cntr=0.3,0.1

Type RM Length L Ch R = 1 ,8508    ,107.7,112.4,117.1
XS GIS Cut Line= 2
2344213.56328693 701683.195745732344109.55053341701986.566276825
#Sta/Elev= 30
       0 2579.43     6.3 2578.97    14.8 2577.03    27.5 2575.53    40.2 2571.96
    48.6 2572.82    57.1 2572.15      74 2566.45    82.4 2562.72     112 2552.29
   116.3 2551.24   133.2 2543.54   152.3 2538.19   158.6 2537.47     167 2537.42
  172.312538.197   179.7 2541.48   185.3 2542.76   192.4 2546.99   197.9 2549.21
   204.2  2550.9   213.6 2551.54   230.4 2550.43   251.6 2553.62   255.8 2556.16
     277 2571.94   289.6 2578.81   298.1 2584.94   308.1 2590.42   320.7 2598.37
#Mann= 3 ,-1,0
       0      .1       0   152.3    .045       0  172.31      .1       0
Bank Sta=152.3,172.31
XS Rating Curve= 0 ,0
Exp/Cntr(USF)=0,0
Exp/Cntr=0.3,0.1

Type RM Length L Ch R = 1 ,8396    ,158.6,156.2,154.5
XS GIS Cut Line= 2
2344204.89555747701679.7286539462343931.86207948 701881.68675036
#Sta/Elev= 30
       0 2578.53    10.8 2577.31    30.2  2573.8    44.5  2572.1    58.8 2569.62
    70.2 2568.52    85.5 2565.74   105.4 2559.76   127.4 2549.34   143.7 2540.73
   153.1 2536.13     156 2535.25   163.9 2534.65   170.6 2533.09     176 2532.48
     185 2533.08   190.8 2535.28   204.6    2539   219.8  2542.4   224.8 2542.83
   239.7 2542.72   249.7 2543.53   259.6 2542.98   264.6 2543.08   270.4 2544.02
   273.2 2544.92   281.8 2548.73   299.4 2557.46   316.1 2566.81   339.6 2577.58
#Mann= 3 ,-1,0
       0      .1       0   170.6    .045       0     185      .1       0
Bank Sta=170.6,185
XS Rating Curve= 0 ,0
Exp/Cntr(USF)=0,0
Exp/Cntr=0.3,0.1

Type RM Length L Ch R = 1 ,8240    ,146.6,145.8,144.3
XS GIS Cut Line= 4
2344084.41411798701567.0481709682343986.46877508701634.656460755
2343919.72725824701738.6692142732343898.92470754701855.683561981
#Sta/Elev= 30
       0 2572.16    17.8 2567.19    34.3 2564.04    53.8 2558.89    76.5 2551.77
    82.9 2549.15    95.3 2542.69   108.1 2538.33   125.4 2529.69   136.3 2524.99
     141 2523.79   153.92522.193   157.2 2521.97   164.8 2522.16   174.3 2522.74
   189.9 2529.57   197.3 2531.46   206.5 2531.56   221.8 2528.73   241.2 2529.14
   244.4 2530.44   257.3 2538.45   269.5 2542.73   285.7 2550.52   293.9 2551.85
   306.1 2556.88   318.3 2560.88   326.4  2562.8   347.9 2570.07   361.4 2573.68
#Mann= 3 ,-1,0
       0      .1       0   153.9    .045       0   164.8      .1       0
Bank Sta=153.9,164.8
XS Rating Curve= 0 ,0
Exp/Cntr(USF)=0,0
Exp/Cntr=0.3,0.1

Type RM Length L Ch R = 1 ,8094    ,89.8,86,83
XS GIS Cut Line= 3
2343969.13331616701459.5683256662343884.18956745701526.309842507
2343757.64071734701748.203716679
#Sta/Elev= 30
       0 2574.29    18.9 2568.35    31.7    2563    67.4 2549.62      73  2545.9
    80.3 2542.79    99.7 2532.76     108 2529.62   118.9 2526.47   129.7 2524.63
   142.4 2516.74   155.8 2513.18   166.6 2512.52   171.2 2512.55  173.812513.198
   180.5 2516.35     185 2517.72   198.8  2519.2   212.6 2518.41   221.8 2519.28
   233.6 2519.35   249.5 2521.07   263.3 2519.88   281.7    2521     292 2519.66
   304.7 2521.48   309.3 2522.91   313.9 2526.31   318.5 2528.65   363.5 2547.53
#Mann= 3 ,-1,0
       0      .1       0   155.8    .045       0  173.81      .1       0
Bank Sta=155.8,173.81
XS Rating Curve= 0 ,0
Exp/Cntr(USF)=0,0
Exp/Cntr=0.3,0.1

Type RM Length L Ch R = 1 ,8008    ,108.3,109,109.6
XS GIS Cut Line= 3
2343887.27142682701401.7834626012343780.36943015701492.313081403
2343748.20252304701750.033570676
#Sta/Elev= 30
       0 2570.56    10.3    2567    35.5 2556.15    84.1 2537.85   101.1 2532.02
   135.1 2523.21     145 2519.44   176.9 2515.39   193.4 2512.09  201.052508.055
   206.2 2507.28   214.6 2508.03   229.6 2513.34   233.7  2514.1   241.7  2514.6
   253.8 2514.43     270 2518.42   280.8 2518.12   294.1 2515.29   298.2 2515.02
   310.3 2516.38   318.3 2518.69   326.4 2521.96   338.5 2523.29   346.5 2528.02
   354.6  2531.8   362.7 2536.63   370.7 2539.06   382.8 2545.02   399.8 2550.65
#Mann= 3 ,-1,0
       0      .1       0  201.05    .045       0   214.6      .1       0
Bank Sta=201.05,214.6
XS Rating Curve= 0 ,0
Exp/Cntr(USF)=0,0
Exp/Cntr=0.3,0.1

Type RM Length L Ch R = 1 ,7899    ,130,134.7,139.4
XS GIS Cut Line= 3
2343793.85256486701329.5523837692343685.02440609701435.491299389
2343633.40326175701712.088177263
#Sta/Elev= 30
       0 2558.25     6.6 2556.48    24.7  2549.1    35.8 2546.21      47 2541.39
    74.9 2532.24   119.6  2520.2   128.2  2516.3   153.6 2508.08   169.9 2506.44
   182.1 2506.69   198.4 2503.85   215.8 2507.21   222.8 2507.56   230.9 2506.06
   243.1 2505.72   254.42501.414   263.5 2500.74   274.6  2501.3   279.7  2502.9
     296 2514.13   304.1 2516.53   311.8 2520.29   320.4 2522.04   332.6 2522.71
   361.1 2526.56   377.4 2529.79   414.7 2544.62   422.2 2548.38   433.2 2551.33
#Mann= 3 ,-1,0
       0      .1       0   254.4    .045       0   274.6      .1       0
Bank Sta=254.4,274.6
XS Rating Curve= 0 ,0
Exp/Cntr(USF)=0,0
Exp/Cntr=0.3,0.1

Type RM Length L Ch R = 1 ,7764    ,216,210.5,205.9
XS GIS Cut Line= 2
2343726.43689129701272.730601754 2343426.9186844701620.402861199
#Sta/Elev= 30
       0 2547.39    40.2  2534.4    53.4 2531.02    85.1 2524.38   101.2 2522.25
   127.3 2515.12   150.5 2509.64   175.1 2506.75   187.3 2503.83   201.2 2497.78
   206.1 2496.48   211.8 2495.88     226 2496.28   238.2  2494.5     254 2495.46
  268.162491.058   274.2 2490.44  282.112491.073   296.3  2492.9   302.6 2495.06
     316 2497.16   327.9 2503.29   333.8 2505.56   345.1  2505.8   359.6 2507.47
   370.2  2507.6   380.7 2510.25   391.3 2511.85   417.7 2519.41   458.9 2532.88
#Mann= 3 ,-1,0
       0      .1       0  268.16    .045       0  282.11      .1       0
Bank Sta=268.16,282.11
XS Rating Curve= 0 ,0
Exp/Cntr(USF)=0,0
Exp/Cntr=0.3,0.1

Type RM Length L Ch R = 1 ,7554    ,199.5,204.2,214.1
XS GIS Cut Line= 3
2343604.77815576  701181.23790192343444.90670128701236.133521813
2343408.30962134 701612.69821279
#Sta/Elev= 30
       0 2537.62     9.9 2535.64    31.9 2528.88    73.7 2519.42    89.5 2517.07
   131.7 2513.52   152.9 2510.44   182.1 2509.28   198.2  2507.4   206.3 2504.08
   226.3 2492.87   234.4 2490.51   242.4 2489.69   258.5 2480.19     2662478.662
   274.6 2477.64   281.82478.938   286.6 2481.32   290.6 2481.81   311.8 2481.35
   326.8 2482.74   338.9 2488.91   346.9 2490.66   375.8 2490.04   403.2 2492.02
   419.3 2494.31   427.3 2497.51   443.4 2499.96   507.7  2516.5   547.4 2530.41
#Mann= 3 ,-1,0
       0      .1       0     266    .045       0   281.8      .1       0
Bank Sta=266,281.8
XS Rating Curve= 0 ,0
Exp/Cntr(USF)=0,0
Exp/Cntr=0.3,0.1
